HEC-RAS study DEERCK.prj: DEERCK

--- DEERCK.g01 (geometry) --- (continued)

Type RM Length L Ch R = 1 ,72800   ,399.8,375.9,351
XS GIS Cut Line= 2
2310181.16260899537456.4209463432309641.87147602537908.865195556
#Sta/Elev= 30
       0 2644.06     107 2643.63   123.3 2642.67   156.8 2638.87   169.2 2638.42
   210.1 2639.09   241.5 2637.12  254.67 2635.25   262.4  2633.5   276.6 2633.33
   287.72635.158   304.1 2636.41   312.4 2635.94   330.2 2637.23     359 2636.98
   381.7 2638.19     419 2637.34   480.4 2637.24   511.5 2636.23   523.7 2636.86
   554.7 2640.81   596.5  2641.9   612.2 2643.76   622.6 2643.89   628.7 2643.31
   640.1 2644.22   648.6 2645.75   664.4  2650.4   685.5  2655.3   703.9 2658.41
#Mann= 5 ,-1,0
       0     .05       0  254.67    .045       0   287.7     .05       0
     380     .07       0     640     .08       0
#XS Ineff= 2 , 0
          162.13 2642.37
Permanent Ineff=
       F       F
Bank Sta=254.67,287.7
XS Rating Curve= 0 ,0
Exp/Cntr(USF)=0,0
Exp/Cntr=0.3,0.1

Type RM Length L Ch R = 1 ,72424   ,322.9,365.8,413.5
XS GIS Cut Line= 4
2309763.73726451537184.6742455772309651.67676935537358.368013077
2309588.64274082 537667.935130962309445.76560949537786.999407069
#Sta/Elev= 30
       0 2641.04    19.6 2640.52    57.7    2641    89.7 2638.73   138.9 2637.63
   204.4 2638.65   221.8 2637.38   258.6 2638.21     279 2638.07   299.4 2635.73
   364.7 2637.25   385.1  2636.5   397.3 2633.59   412.2 2632.16   425.9 2632.76
   431.72633.541   438.2 2634.71   466.7 2637.13   491.2  2641.9   546.6 2642.33
   560.8 2643.11   568.3 2643.01   575.3 2642.01   593.3 2642.63   603.4  2643.9
   611.9 2646.27   626.1 2652.34   654.5 2666.47   684.6 2682.78   708.6 2694.59
#Mann= 4 ,-1,0
       0     .05       0   397.3    .045       0   431.7     .05       0
  592.62      .1       0
#XS Ineff= 2 , 0
          156.81 2645.02
Permanent Ineff=
       F       F
Bank Sta=397.3,431.7
XS Rating Curve= 0 ,0
Exp/Cntr(USF)=0,0
Exp/Cntr=0.3,0.1

Type RM Length L Ch R = 1 ,72058   ,305.5,287.3,268.3
XS GIS Cut Line= 4
2309718.53595947537119.3708857052309522.30054931537273.242097672
2309334.06595645537312.708824076 2309212.5468073 537680.98436774
#Sta/Elev= 30
       0 2641.27   113.1 2640.39     154 2636.94   213.8 2637.14   255.6 2638.01
   274.8  2637.4   296.5  2635.7     321 2636.22   346.52635.248   353.7 2633.11
   357.8  2631.3     366 2630.38   382.3 2630.72   386.4 2631.28   390.5 2632.95
   394.6 2634.65   406.8 2635.23     428 2638.24   439.5    2639   456.2  2638.9
   467.5 2641.23   494.2 2649.41   505.4 2651.68     518 2653.16   631.7 2660.14
   648.6 2661.82   720.2 2672.92   762.3  2681.1   791.9 2686.72   829.5 2692.21
#Mann= 5 ,-1,0
       0     .05       0   346.5     .05       0   353.7    .045       0
   390.5     .05       0   762.3      .1       0
Bank Sta=353.7,390.5
XS Rating Curve= 0 ,0
Exp/Cntr(USF)=0,0
Exp/Cntr=0.3,0.1

Type RM Length L Ch R = 1 ,71771   ,444.9,432,418.4
XS GIS Cut Line= 3
2309645.71159696536768.0413077162309185.73882994537130.173514508
2309202.87541143537683.114542243
#Sta/Elev= 30
       0 2639.37    83.4  2638.7   134.3 2640.14   202.3  2638.3   292.1  2638.5
   320.9 2636.63     343 2633.27     394 2633.54     4012631.041   404.1 2630.03
   422.2 2629.54   434.7 2629.95   437.82631.023   440.6 2631.95   451.9 2635.09
   521.2 2634.47   570.9 2635.29     583 2636.26   664.5 2636.38   692.5 2635.48
   708.5 2638.62   724.5  2639.9   740.5 2647.12   756.5 2651.33   924.7 2658.22
   964.6  2660.7  1007.3 2665.92  1052.6 2673.62  1075.9  2678.7  1138.6 2691.25
#Mann= 7 ,-1,0
       0     .05       0   320.9     .07       0     401    .045       0
   437.8     .07       0   440.6     .08       0   570.9     .05       0
  1075.9      .1       0
Bank Sta=401,437.8
XS Rating Curve= 0 ,0
Exp/Cntr(USF)=0,0
Exp/Cntr=0.3,0.1

Type RM Length L Ch R = 1 ,71339   ,399.7,416.7,423
XS GIS Cut Line= 3
2309419.03538587536193.4434702932308981.49758306536873.472103574
2308512.33054149537208.214880421
#Sta/Elev= 30
       0 2636.94   108.8 2634.78   302.9 2636.54   323.1 2631.88   356.4  2629.5
   389.7 2632.66   475.3 2632.78   508.4 2630.76   560.9 2632.95     580 2632.56
   598.1 2628.92   608.5 2627.24   624.1 2628.93   638.6 2633.94   765.5  2631.2
   808.6 2633.31   820.8 2631.29   849.4 2633.25  1035.4 2632.19  1093.3 2634.28
  1111.2 2631.69  1124.7 2633.56  1150.6  2632.3  1247.6 2634.95  1267.2 2645.25
    1282  2647.5  1301.6 2663.09  1326.2 2675.55  1350.8    2683    1385 2688.44
#Mann= 5 ,-1,0
       0     .05       0     410     .07       0   598.1    .045       0
   624.1     .08       0 1268.63      .1       0
#XS Ineff= 2 , 0
                          960.84         2640.75
Permanent Ineff=
       F       F
Bank Sta=598.1,624.1
XS Rating Curve= 0 ,0
Exp/Cntr(USF)=0,0
Exp/Cntr=0.3,0.1

Type RM Length L Ch R = 1 ,70922   ,347.8,377.4,403.1
XS GIS Cut Line= 3
2309380.66385901536053.2735863772308998.50358173536318.010314772
2308236.31800079536986.257056608
#Sta/Elev= 30
       0 2654.16    29.8 2640.51    83.6 2635.56   217.6 2634.02   474.5 2636.26
   519.8 2631.87   615.3 2631.69   638.9 2629.04   651.7 2630.41   774.9 2630.62
   803.4 2628.08   819.1 2626.42   837.3 2628.13   845.8 2632.03   864.1 2629.83
   936.1 2630.63     949 2628.97   961.2 2631.99   973.8 2632.57  1175.5 2632.09
  1222.8 2633.63  1248.3 2648.79  1265.9  2650.9  1281.9 2664.44  1333.3 2696.57
  1384.3 2719.83  1420.2 2732.85  1446.8 2739.86  1460.9 2742.03  1478.5    2740
#Mann= 6 ,-1,0
       0     .05       0     340     .07       0   494.9     .08       0
   803.4    .045       0   837.3     .08       0   854.9      .1       0
#XS Ineff= 2 , 0
                         1037.47         2646.28
Permanent Ineff=
       F       F
Bank Sta=803.4,837.3
XS Rating Curve= 0 ,0
Exp/Cntr(USF)=0,0
Exp/Cntr=0.3,0.1

Type RM Length L Ch R = 1 ,70545   ,500.4,504.5,507.3
XS GIS Cut Line= 4
2309368.95575783536053.7476657822308963.04719378536317.324655425
2308272.47548091536288.3311865652308074.79273868536512.371627762
#Sta/Elev= 30
       0 2649.73    13.6 2641.94    20.4 2640.08    86.9 2635.06   220.3    2634
   471.5 2635.85   506.9 2631.76     651 2630.48   662.3 2628.32   835.2 2629.73
   871.2 2629.28  876.43 2627.51   883.2 2625.41   899.2 2625.65  906.34 2627.49
   919.2 2632.19   943.3 2634.34  1035.3 2634.62  1063.2 2636.86  1175.2 2640.08
  1187.3 2642.83  1198.6 2649.41  1205.8  2651.5  1255.3 2654.64    1261 2660.76
    1267 2672.62  1326.2 2689.25  1381.2 2702.11    1427 2705.86  1473.9 2701.89
#Mann= 6 ,-1,0
       0     .05       0     340     .07       0  643.98     .08       0
  843.98      .1       0  876.43    .045       0  906.34      .1       0
Bank Sta=876.43,906.34
XS Rating Curve= 0 ,0
Exp/Cntr(USF)=0,0
Exp/Cntr=0.3,0.1

Type RM Length L Ch R = 1 ,70040   ,410.3,407.6,403.8
XS GIS Cut Line= 2
2309280.32009906535901.6904596352308155.18900338535758.647227357
#Sta/Elev= 30
       0 2636.94     101 2636.26   209.8 2632.27   262.2 2633.51   286.4 2629.88
   322.9 2628.44   379.8 2629.56   403.4 2627.26     480 2626.37     480 2626.38
   508.2 2628.06   592.9 2628.54     605 2626.85  611.09 2624.06   617.1 2623.19
   629.2 2624.04   653.4 2625.45   673.5 2623.47   694.6 2628.42   754.2 2626.69
   769.7 2630.39   790.5 2632.16   898.5 2632.23  1040.5 2636.78  1060.6 2639.58
  1076.7  2648.8  1088.8 2650.58  1100.9 2662.23    1113 2671.42  1134.2 2683.18
#Mann= 11 ,-1,0
       0     .05       0     380     .08       0     480     .07       0
     500      .1       0     580     .08       0  611.09    .045       0
   629.2     .08       0     780      .1       0     880     .07       0
     980      .1       0    1080     .08       0
#XS Ineff= 2 , 0
          376.92 2633.32
Permanent Ineff=
       F       F
Bank Sta=611.09,629.2
XS Rating Curve= 0 ,0
Exp/Cntr(USF)=0,0
Exp/Cntr=0.3,0.1

Type RM Length L Ch R = 1 ,69632   ,804.7,782,751
XS GIS Cut Line= 2
2309301.66983522535457.6159474882308165.86387146535427.726316863
#Sta/Elev= 30
       0 2633.89   243.6 2633.88   305.6 2631.69   437.6 2631.99   461.7 2630.59
   469.7 2628.88   481.7 2623.83   501.7 2626.39   509.7 2625.12   533.7 2625.96
  545.06 2623.19   553.7 2622.16   570.82623.221   581.7 2626.61   613.7 2624.99
   625.7 2625.84   645.7 2624.82   661.7 2626.92   729.7 2626.19     786 2628.22
   873.8 2627.84  1025.8 2632.27  1033.9 2634.16  1041.9    2639  1053.9 2639.62
  1057.9  2641.4  1065.9 2647.53  1109.1 2670.04  1120.8 2675.04  1136.2 2679.86
#Mann= 9 ,-1,0
       0     .05       0     400     .08       0  545.06    .045       0
   570.8     .08       0     700     .07       0     790      .1       0
     890     .07       0     990     .05       0    1090     .08       0
Bank Sta=545.06,570.8
XS Rating Curve= 0 ,0
Exp/Cntr(USF)=0,0
Exp/Cntr=0.3,0.1

Type RM Length L Ch R = 1 ,68850   ,345,379.9,390.1
XS GIS Cut Line= 4
2309536.51693299534793.6391528842308829.84066606534814.988889045
2308526.67441258535088.2655119052308112.48953106535126.695036994
#Sta/Elev= 30
       0 2637.35   140.4  2632.1   220.4 2634.84   648.7 2632.87   734.2 2630.98
   757.7 2626.83   774.9 2626.28     806 2622.32   841.7 2622.82   854.6 2624.89
   895.5 2624.11   905.2 2621.13   919.3 2622.43   935.4 2620.04     9542622.255
   967.2 2623.51   989.3 2621.52  1004.3 2623.68    1027 2623.81  1055.3 2621.88
  1080.7 2625.91  1226.1  2625.3  1310.5 2629.83    1423 2629.77  1430.8 2631.96
    1439 2636.92  1451.1 2638.23  1467.2 2649.61  1491.3 2662.63  1531.1 2679.17
#Mann= 10 ,-1,0
       0     .05       0     777      .1       0     917     .05       0
   919.3    .045       0     954     .05       0    1007      .1       0
    1067     .05       0 1135.15      .1       0 1235.15     .05       0
 1435.15      .1       0
Bank Sta=919.3,954
XS Rating Curve= 0 ,0
Exp/Cntr(USF)=0,0
Exp/Cntr=0.3,0.1

Type RM Length L Ch R = 1 ,68471   ,539.3,548.5,542.1
XS GIS Cut Line= 5
2309504.98264877534743.0330390982308842.83958156534750.765987039
2308734.29217171534651.4032107142308676.53571165534656.653797993
2308037.78083476534860.113711454
#Sta/Elev= 30
       0 2639.04    56.8 2632.83   161.1 2631.04   204.6 2631.98   232.3 2635.09
   249.6 2635.31   789.8  2631.6     824 2628.34   831.6 2625.06   838.12619.599
   843.6 2618.14   855.7 2618.24   860.8 2619.67   867.7 2621.48   925.4 2622.71
   985.3 2621.25   993.7 2623.01  1062.3 2623.43  1123.8 2621.54  1136.4  2623.3
    1170 2622.07  1189.6 2625.25  1241.3  2624.6  1272.4 2627.78  1388.3 2629.34
  1400.9 2633.94  1417.7 2635.24  1433.8 2644.97    1473 2660.23  1537.7 2690.37
#Mann= 4 ,-1,0
       0     .05       0  712.19      .1       0   838.1    .045       0
   860.8      .1       0
Bank Sta=838.1,860.8
XS Rating Curve= 0 ,0
Exp/Cntr(USF)=0,0
Exp/Cntr=0.3,0.1

Type RM Length L Ch R = 1 ,67922   ,146.7,151.3,155.9
XS GIS Cut Line= 4
 2309034.6705805534183.5577792522308579.65679172534259.820414091
2308142.28845605534319.3035653432307981.41795086534342.345864809
#Sta/Elev= 30
       0  2635.9   205.3 2633.65   233.7 2631.84   274.3 2630.97   318.9 2631.98
   375.7 2631.41   391.9 2630.04   420.3 2624.62   485.1 2624.86   513.3 2620.49
   569.8 2620.94   577.9 2617.71     590 2616.75   604.2 2617.42   614.2 2618.59
   626.3 2617.13   638.5  2618.7   650.4  2623.2   658.6 2624.27   670.8 2622.28
   751.5 2621.48   783.8 2624.69   816.1 2624.66   852.4 2629.51     861 2631.31
   876.6 2636.76     917 2654.89   973.4 2675.04   997.8 2681.36  1065.3 2691.73
#Mann= 6 ,-1,0
       0     .05       0  501.36     .08       0   577.9     .04       0
   604.2     .08       0  731.36     .05       0  831.36      .1       0
Bank Sta=577.9,604.2
XS Rating Curve= 0 ,0
Exp/Cntr(USF)=0,0
Exp/Cntr=0.3,0.1

Type RM Length L Ch R = 1 ,67771   ,361.7,344.9,327.3
XS GIS Cut Line= 2
2309022.69151477534123.7386067742307893.54112414534130.520290801
#Sta/Elev= 30
       0 2634.54    82.5 2632.41   118.5 2633.16   158.5 2632.16   198.8 2632.84
   270.5 2632.16   334.5 2622.92   434.5 2624.44   475.9 2622.62   526.5 2623.49
   540.3  2618.7   546.5 2616.56   556.4 2616.55   582.5 2616.64   590.5 2618.53
   598.5 2620.67   610.5 2620.47   626.5 2622.03   682.5 2620.69   698.5 2622.92
   735.6 2623.59   794.5 2621.62   834.5 2623.94   862.8 2630.49   874.5 2635.39
   914.5 2655.35  1006.5 2690.06  1054.5 2700.67  1111.8 2709.74  1129.2 2711.45
#Mann= 4 ,-1,0
       0     .05       0   540.3     .04       0   590.5     .05       0
    1010      .1       0
#XS Ineff= 2 , 0
          508.31 2635.13
Permanent Ineff=
       F       F
Bank Sta=540.3,590.5
XS Rating Curve= 0 ,0
Exp/Cntr(USF)=0,0
Minor Loss Coefficient=0
Exp/Cntr=0.3,0.1

Type RM Length L Ch R = 1 ,67426   ,289.6,293.1,319
XS GIS Cut Line= 4
2308795.69432056533755.2915357812308542.45926713533736.674478512
2308189.34858123533860.6556826532307890.45227498533899.085207743
#Sta/Elev= 30
       0 2632.22    31.6 2632.47    51.7 2631.44    83.7  2624.1   111.8 2626.05
   135.9 2626.28   204.1 2623.97   236.2 2620.27   240.2 2620.16   252.2 2623.07
   260.6 2621.46   294.5 2622.09   312.6 2620.54   366.6 2620.99   394.2 2619.14
   400.3 2617.49     413 2616.47   459.8  2616.6   465.5 2617.47   476.8 2620.61
   527.7 2618.77   536.1 2619.55   544.6 2621.84   570.1 2621.19   612.4 2622.71
     706  2620.8   794.1  2624.5   843.1 2629.65     912 2644.45   929.5 2647.31
#Mann= 5 ,-1,0
       0     .05       0  393.92     .07       0   400.3     .04       0
   465.5     .07       0  503.92     .05       0
#XS Ineff= 2 , 0
          247.51 2627.27
Permanent Ineff=
       F       F
Bank Sta=400.3,465.5
XS Rating Curve= 0 ,0
Exp/Cntr(USF)=0,0
Exp/Cntr=0.3,0.1

Type RM Length L Ch R = 1 ,67133   ,283,281.1,274.9
XS GIS Cut Line= 2
2308533.07933343533506.2500623832307815.72819842533756.041975465
#Sta/Elev= 30
       0 2627.74    13.7 2624.77    22.1 2624.21      25 2623.39    34.8 2617.36
    37.6  2616.5    43.3 2615.81    62.7 2616.44      69 2617.04    84.7 2616.91
    94.1 2617.66   153.8 2618.93   161.9 2618.72   170.4 2617.11   178.9 2616.37
   212.7 2618.47   221.2 2619.76   288.7 2618.34   310.2 2618.29   318.6  2619.1
   382.2  2617.7   386.4 2618.05   394.9 2620.34   398.9 2620.55   475.3 2619.84
   530.4 2621.28   580.6 2621.36   621.9 2624.11   682.9 2623.59   759.6 2625.15
#Mann= 5 ,-1,0
       0     .05       0    37.6     .04       0    62.7     .05       0
     220     .07       0     340     .05       0
#XS Ineff= 2 , 0
                          527.57         2623.63
Permanent Ineff=
       F       F
Bank Sta=37.6,62.7
XS Rating Curve= 0 ,0
Exp/Cntr(USF)=0,0
Exp/Cntr=0.3,0.1

Type RM Length L Ch R = 1 ,66852   ,509.5,516.8,512.8
XS GIS Cut Line= 4
2308593.01550751533289.0186559432308415.52202631533265.962300875
2308037.76545449533463.5505900612307698.30464953533621.538637651
#Sta/Elev= 30
       0    2629    33.1 2627.65    69.4 2624.79   117.8 2623.16   170.3 2623.76
   174.3 2622.71   209.8 2622.16   269.8 2623.15   272.8  2622.7   278.7 2617.06
   282.22614.734   290.5 2613.91   313.7 2614.73   340.9 2618.78   358.8 2619.63
   376.5 2619.02   410.3 2618.57   503.9 2617.02   552.9 2617.96   561.9 2619.12
     578 2618.85   595.7 2620.25   622.8 2620.14   642.3 2618.81   661.9 2620.07
   752.2 2619.63   765.9 2620.04   789.3 2622.41   862.9  2622.7   979.7 2624.08
#Mann= 8 ,-1,0
       0     .07       0    33.1     .05       0   170.3     .07       0
   282.2     .04       0   313.7     .05       0   376.5     .07       0
   410.3     .05       0   862.9      .1       0
#XS Ineff= 1 ,-1
  609.78  938.35 2623.24
Permanent Ineff=
       F
Bank Sta=282.2,313.7
XS Rating Curve= 0 ,0
Exp/Cntr(USF)=0,0
Exp/Cntr=0.3,0.1

Type RM Length L Ch R = 1 ,66335   ,298.1,302.7,305.5
XS GIS Cut Line= 2
2308294.23801303532908.6884113422307481.48934677533417.533176583
#Sta/Elev= 30
       0 2622.03    31.1 2622.75   125.1 2620.76   204.4 2622.78   224.2 2622.29
   243.1 2618.66     262 2617.98   272.3 2618.91   290.3 2617.91   338.5 2617.86
   361.1 2618.86   384.7 2615.86     414 2617.44   441.3 2616.74   460.52614.787
   468.3  2614.5   477.8 2612.87   490.9 2612.59     498 2612.71   503.9 2614.48
   512.1 2616.46     521  2616.6     533 2617.84   587.6 2617.95   602.6 2619.57
   669.4 2619.47   704.2  2622.1   823.6 2623.09   905.5 2621.61   958.9 2621.86
#Mann= 6 ,-1,0
       0     .05       0   441.3     .07       0   460.5     .04       0
   468.3     .04       0   503.9     .07       0     521     .05       0
Bank Sta=468.3,503.9
XS Rating Curve= 0 ,0
Exp/Cntr(USF)=0,0
Exp/Cntr=0.3,0.1

Type RM Length L Ch R = 1 ,66032   ,501.5,495.4,487.3
XS GIS Cut Line= 3
2308155.18900338532694.9600882692307474.13241985533034.420893227
2307339.62908203533337.587146712
#Sta/Elev= 30
       0 2621.97   147.1 2622.11   186.6 2620.77   213.4 2622.93   239.5 2623.03
   251.3 2621.85   269.4  2617.9   281.3 2616.88   373.8 2617.32   388.7    2614
   423.5 2614.45   433.4 2612.64   441.4  2612.2   454.8 2612.24  461.33 2614.52
   463.7 2615.53   468.2 2615.71   503.9 2614.07   521.8 2618.07   539.7 2615.32
   579.9 2616.67   602.3 2615.28   611.2 2615.59   624.6 2617.82   657.1 2618.69
   785.9 2619.12   816.5 2620.31   895.3 2619.62   946.4  2620.7  1092.6 2621.57
#Mann= 6 ,-1,0
       0     .05       0     380     .07       0   423.5     .04       0
  461.33     .05       0     490     .07       0     600     .05       0
#XS Ineff= 2 , 0
          295.02 2619.79
Permanent Ineff=
       F       F
Bank Sta=423.5,461.33
XS Rating Curve= 0 ,0
Exp/Cntr(USF)=0,0
Exp/Cntr=0.3,0.1

Type RM Length L Ch R = 1 ,65537   ,519.8,527.1,518.5
XS GIS Cut Line= 2
 2307879.7774069532227.4008663452306921.17425328532957.561843048
#Sta/Elev= 30
       0 2621.11   291.1  2621.5   323.5 2619.22     333 2616.33   351.5 2612.99
   366.6 2613.75   386.7  2613.5   426.9 2611.98     432 2611.22     442 2610.98
   457.7 2611.08  462.94 2612.04   469.1 2615.22   478.2 2615.71   500.5 2614.96
   543.3 2614.96   577.3 2614.19   602.9 2615.55     628 2612.69   658.2 2612.52
   663.2 2612.76   678.3  2615.6   743.7 2614.86     783 2617.62   839.2 2617.19
   857.2 2615.77   868.7 2615.58   905.8 2616.92   974.3 2616.45    1205 2620.71
#Mann= 5 ,-1,0
       0     .05       0   426.9     .04       0  462.94     .05       0
     570     .03       0     690     .05       0
#XS Ineff= 2 , 0
                          795.35         2618.37
Permanent Ineff=
       F       F
Bank Sta=426.9,462.94
XS Rating Curve= 0 ,0
Exp/Cntr(USF)=0,0
Exp/Cntr=0.3,0.1

Type RM Length L Ch R = 1 ,65010   ,164.2,160.1,159.3
XS GIS Cut Line= 2
2307546.72152279531984.0138741112306803.75070439532665.070457643
#Sta/Elev= 30
       0 2620.41    52.3 2619.33   144.2 2619.31     181 2617.21   238.5 2617.38
   248.9  2616.8   263.9 2614.44   301.9 2614.58   321.4 2614.52   356.9 2613.85
   398.3 2614.99   432.1 2612.95   439.8  2612.7   451.6 2610.75   475.4 2608.84
   483.9 2609.25  487.73 2610.82     493  2613.9   510.8 2614.03   534.5 2612.56
   551.9  2614.9   567.8 2613.95   589.5 2614.29   616.6 2612.18   650.9 2613.94
   712.1 2614.08     767 2615.22   809.5 2614.84   882.5 2617.84  1007.9 2618.94
#Mann= 6 ,-1,0
       0     .05       0   301.9     .03       0   321.4     .05       0
   432.1     .03       0   451.6     .04       0  487.73     .05       0
#XS Ineff= 2 , 0
                          710.65            2618
Permanent Ineff=
       F       F
Bank Sta=451.6,487.73
XS Rating Curve= 0 ,0
Exp/Cntr(USF)=0,0
Exp/Cntr=0.5,0.3

Type RM Length L Ch R = 1 ,64849   ,70.9,65.7,66
XS GIS Cut Line= 2
2307435.70289475531845.2405890652306701.27197082532575.401565768
#Sta/Elev= 30
       0 2618.75    28.3 2618.45    61.8 2615.76   112.1 2616.46   153.1 2614.88
   268.3 2616.52   283.6 2616.24   303.9 2613.81   360.3 2614.89   402.7 2614.61
   419.7 2613.39   453.8 2613.74   466.3 2612.99   480.5 2609.75   493.5 2608.11
   510.5 2608.15  521.47 2609.72     537 2611.67   556.8  2611.6     571 2613.33
   582.3 2612.27   597.2 2613.59   614.1 2613.39   633.2 2615.42   650.2 2615.15
     710 2615.54   856.7 2615.31     868 2613.44   918.9 2617.59  1035.6  2617.8
#Mann= 6 ,-1,0
       0     .06       0   480.5     .04       0  521.47     .05       0
     571     .06       0   650.2     .05       0     710     .06       0
#XS Ineff= 5 ,-1
   27.91  261.13 2618.42  261.13     420  2614.8   535.9  701.42  2615.5
  701.42  920.28 2617.26  920.28  1035.6  2615.5
Permanent Ineff=
       F       F       F       F       F
Bank Sta=480.5,521.47
XS Rating Curve= 0 ,0
Exp/Cntr(USF)=0,0
Exp/Cntr=0.5,0.3

Type RM Length L Ch R = 1 ,64784   ,234.1,225.5,213.1
XS GIS Cut Line= 2
2307395.13839605531798.2711695112306660.70747211532528.432146214
#Sta/Elev= 30
       0 2618.58    18.3 2618.43    60.6 2618.19   122.6 2615.01   230.4 2615.44
   291.8 2615.56   303.1  2615.7   327.5 2613.68   370.8 2613.17   431.2 2613.64
   483.6 2613.76   520.4 2609.89   526.1 2608.33   533.1 2608.02   548.8 2609.84
   577.1 2613.22   599.8 2612.47   622.5 2615.44   650.9 2615.33   711.3 2615.25
   790.5 2614.34   844.2 2614.96   850.2 2613.95   858.3 2613.27   869.7 2614.74
     901 2615.02   917.5 2617.81   931.9 2618.44   991.3 2618.97  1035.6 2619.31
#Mann= 14 ,-1,0
       0     .05       0    18.3     .06       0   230.4     .05       0
   291.8     .06       0   370.8     .07       0   431.2     .06       0
   520.4     .04       0   548.8     .06       0   650.9     .05       0
   711.3     .06       0   790.5     .05       0   850.2     .06       0
   931.9     .05       0   991.3     .06       0
#XS Ineff= 4 ,-1
       0   491.7  2614.3   568.3  697.15  2615.5  697.15  937.37 2616.83
  937.37  1035.6  2615.5
Permanent Ineff=
       F       F       F       F
Bank Sta=520.4,548.8
XS Rating Curve= 0 ,0
Exp/Cntr(USF)=0,0
Exp/Cntr=0.5,0.3

Type RM Length L Ch R = 1 ,64558   ,444.9,470.6,492.9
XS GIS Cut Line= 4
2307312.85571693531588.2386147632307108.02312322 531672.33781792
2306844.27100541532024.6963209362306530.47408153532607.426170009
#Sta/Elev= 30
       0 2615.03    74.2 2614.35   227.8 2615.68   281.9 2614.24   513.4 2614.34
   536.2 2612.62     655 2614.36   666.7 2614.12   682.7 2610.85   697.4 2612.11
   711.62609.817     721 2607.78   734.8 2607.82   742.92609.987   748.4 2612.38
   754.6 2613.12   807.5 2611.14   824.4 2612.66   836.2  2611.1   866.6 2612.39
   921.1 2612.33   931.7 2611.34   945.5 2612.93   995.7 2613.25  1016.3 2617.38
  1066.7 2616.54  1193.5 2619.93  1243.7 2622.56    1280 2630.39  1323.4 2633.43
#Mann= 7 ,-1,0
       0     .05       0  671.56     .07       0   711.6     .04       0
   742.9     .07       0  881.56     .05       0 1091.56     .06       0
 1311.56     .05       0
#XS Ineff= 2 , 0
          437.21 2619.49
Permanent Ineff=
       F       F
Bank Sta=711.6,742.9
XS Rating Curve= 0 ,0
Exp/Cntr(USF)=0,0
Exp/Cntr=0.3,0.1

Type RM Length L Ch R = 1 ,64088   ,527.6,578.3,627.6
XS GIS Cut Line= 2
 2307297.3776906531513.0017936222305896.38691755532035.253240897
#Sta/Elev= 30
       0 2615.31   184.8 2614.19   312.9 2614.85   355.7 2614.25   381.2 2611.78
   428.2 2612.15   513.5 2610.89   534.9 2612.54   637.3 2612.02   675.9 2613.04
   682.1 2612.61   694.5 2609.26   701.4 2607.42   709.9 2606.84   735.5 2607.07
   747.4 2609.06   752.6    2611   769.7 2611.12   799.6 2609.31   867.9 2608.75
   884.9 2610.88   906.3 2610.81   918.4 2614.24   931.9 2615.64    1133 2614.57
    1332 2617.16  1358.8 2620.73  1440.9 2644.33    1457 2650.29  1495.2 2668.46
#Mann= 7 ,-1,0
       0     .05       0     490     .07       0     560     .05       0
     600     .07       0   694.5     .04       0   747.4     .07       0
     810     .05       0
Bank Sta=694.5,747.4
XS Rating Curve= 0 ,0
Exp/Cntr(USF)=0,0
Exp/Cntr=0.3,0.1

Type RM Length L Ch R = 1 ,63509   ,740.8,701.9,656.9
XS GIS Cut Line= 4
2307283.32903705531490.8876841912306874.20483372531510.049731339
2306615.02957981531263.288953638 2305816.3913012531561.130951931
#Sta/Elev= 30
       0 2615.34   151.3 2613.84   239.4 2615.19   366.4 2612.93   423.4 2614.05
   448.4 2610.15   495.2 2610.85   499.3 2610.15   506.3 2606.85   511.8 2605.49
   516.3 2605.75   522.8 2607.55   533.3 2606.42   550.1 2605.53   573.3 2606.29
   592.7 2609.68   631.3 2608.04   660.6  2608.3   671.9 2611.09     683 2611.94
   808.9 2610.44   915.6 2612.42   992.5 2611.47  1060.8 2612.73    1112 2611.52
  1163.2 2613.44  1316.9 2612.39  1483.2  2613.1  1551.7 2614.53  1619.8 2620.21
#Mann= 9 ,-1,0
       0     .05       0     350     .07       0     390     .05       0
  419.57     .07       0  459.57     .05       0   533.3     .04       0
   573.3     .08       0  599.57     .07       0  699.57     .05       0
#XS Ineff= 2 , 0
                          771.15         2613.76
Permanent Ineff=
       F       F
Bank Sta=533.3,573.3
XS Rating Curve= 0 ,0
Exp/Cntr(USF)=0,0
Exp/Cntr=0.3,0.1

Type RM Length L Ch R = 1 ,62807   ,369.1,357.1,330.1
XS GIS Cut Line= 4
2307470.51520545531190.770368913 2307214.8455255530961.458387925
2306743.04271404530982.544547095 2305744.0859233 531383.18157135
#Sta/Elev= 30
       0 2619.52   138.7 2619.04   152.9 2617.91   181.2 2614.01   218.1 2612.78
   298.7 2612.28   331.9 2610.25   343.4 2610.36   402.2 2605.77   426.2 2605.03
   466.2 2605.67   518.3 2608.78   575.7 2607.05   646.4 2609.57   670.4 2608.46
   682.4 2609.46   767.3 2608.34   802.6 2610.36   840.4 2609.22   896.8 2610.09
    1023 2609.39  1147.1 2610.01  1193.7 2611.47  1348.6 2611.28  1391.8 2612.75
  1628.7 2611.66  1758.1 2612.18  1861.8 2614.03    1879 2615.84    1892 2618.44
#Mann= 3 ,-1,0
       0     .05       0   402.2     .04       0   466.2     .05       0
#XS Ineff= 2 , 0
                         1066.67         2613.06
Permanent Ineff=
       F       F
Bank Sta=402.2,466.2
XS Rating Curve= 0 ,0
Exp/Cntr(USF)=0,0
Minor Loss Coefficient=0
Exp/Cntr=0.3,0.1

Type RM Length L Ch R = 1 ,62450   ,796.8,793.9,782.3
XS GIS Cut Line= 3
2307405.76054873530280.1467822782307089.46816116530707.141505496
2305639.79471814531210.573555709
#Sta/Elev= 30
       0 2676.35      71  2668.1    90.9 2667.57   177.4 2678.65   199.2 2675.65
   225.3 2668.82   253.5 2658.52   304.9 2632.86   324.8 2625.05     345 2619.88
   385.1 2617.87   583.6 2617.69     609 2608.71   630.1 2609.12   638.6 2606.71
   655.5 2607.43   668.2 2604.99     681  2603.7   719.1 2605.17   727.5 2607.74
   833.4 2607.58   875.7 2610.23  1040.9 2608.65  1135.1 2611.54  1303.4 2609.64
  1391.1 2612.81  1985.1 2612.01  2010.5 2613.48  2026.9 2617.73    2066 2637.56
#Mann= 4 ,-1,0
       0      .1       0     310     .05       0   668.2     .04       0
   719.1     .05       0
#XS Ineff= 2 , 0
                         1169.87         2615.93
Permanent Ineff=
       F       F
Bank Sta=668.2,719.1
XS Rating Curve= 0 ,0
Exp/Cntr(USF)=0,0
Exp/Cntr=0.3,0.1

Type RM Length L Ch R = 1 ,61656   ,730.3,707.3,687.8
XS GIS Cut Line= 2
2307138.26639311529892.7990859332305290.29481507 530840.88885206
#Sta/Elev= 30
       0 2683.73    53.4 2685.15   156.3 2682.77   204.7 2679.71   251.4 2672.46
   281.1  2662.8   317.1  2644.9     353 2604.66   357.5 2603.08   373.2 2602.71
     397 2604.11   408.9 2608.08   438.4 2607.65   459.4 2603.66   478.9 2603.62
   510.4 2604.72   523.9 2607.55   591.3 2605.97   631.7 2609.22   672.2 2607.61
   730.7 2609.27    1021 2608.13  1112.8 2609.88    1369 2610.81  1523.1  2609.3
  1962.9 2609.88    1976 2610.87  1998.6 2616.76  2025.3 2627.43    2077 2651.94
#Mann= 4 ,-1,0
       0      .1       0     353     .04       0     397      .1       0
     530     .05       0
#XS Ineff= 2 , 0
                         1373.68         2619.57
Permanent Ineff=
       F       F
Bank Sta=353,397
XS Rating Curve= 0 ,0
Exp/Cntr(USF)=0,0
Exp/Cntr=0.3,0.1

Type RM Length L Ch R = 1 ,60949   ,242.6,229.8,220
XS GIS Cut Line= 4
2307141.79889168529364.3516796432306476.52912358529407.738838432
2306299.36489186529671.6773877332305153.22078051530626.194881093
#Sta/Elev= 30
       0 2689.74    37.7 2686.96   101.8  2674.1     198 2642.95   242.1 2631.21
   278.2 2625.18   318.4 2621.65   450.6 2619.04   478.6 2614.11   510.7 2611.65
   676.6 2610.79   705.5 2613.24   716.6 2607.69  728.22 2604.76   746.3 2602.43
   757.3 2602.67   763.1 2604.74   769.6  2606.7   861.1 2605.62   904.2 2607.12
   938.2 2605.68   967.1 2607.72  1311.7 2604.95  1354.3 2607.45  1507.7 2606.17
  1597.8 2608.15  2376.7 2608.69  2393.8 2609.81    2415 2615.97  2476.1 2648.31
#Mann= 7 ,-1,0
       0      .1       0     310     .12       0  716.68      .1       0
  728.22     .04       0   763.1      .1       0  836.68     .05       0
 2464.57      .1       0
#XS Ineff= 2 , 0
          693.52 2619.51 1947.37         2621.54
Permanent Ineff=
       F       F
Bank Sta=728.22,763.1
XS Rating Curve= 0 ,0
Exp/Cntr(USF)=0,0
Exp/Cntr=0.3,0.1

Type RM Length L Ch R = 1 ,60719   ,667.6,670,681
XS GIS Cut Line= 3
2306360.83003347528984.7140402392306147.50983609529592.134263286
2305012.21251445530452.646245937
#Sta/Elev= 30
       0 2689.38    98.1 2688.92   217.4 2686.36   243.4 2684.28   263.3 2680.99
   284.5 2674.44   301.5 2665.22   331.2 2643.07   348.1 2626.37   365.1 2612.41
   390.5 2603.98   407.5 2602.06   449.9 2602.16  457.44    2604   466.8 2606.08
   543.1 2604.71   598.3    2607   728.3 2606.25   783.5  2604.4   888.9 2607.46
  1038.1 2605.41  1100.9 2607.28  1149.9 2605.76  1201.8 2607.21  1751.8 2607.16
  1963.1 2608.47    1973 2609.36  1991.7 2616.58  2053.3 2649.84  2068.4 2656.74
#Mann= 10 ,-1,0
       0      .1       0      70     .12       0     180      .1       0
     280     .12       0     340      .1       0   390.5     .04       0
  457.44     .08       0     490     .07       0     590     .05       0
 1883.79      .1       0
#XS Ineff= 2 , 0
                         1536.84         2617.79
Permanent Ineff=
       F       F
Bank Sta=390.5,457.44
XS Rating Curve= 0 ,0
Exp/Cntr(USF)=0,0
Exp/Cntr=0.3,0.1

Type RM Length L Ch R = 1 ,60049   ,980.2,918.1,871.4
XS GIS Cut Line= 4
2305875.64889693528573.9166844222305893.16735685528992.176246792
2305206.43868248529839.6063662032304720.69038131530256.688290156
#Sta/Elev= 30
       0 2681.52    79.3 2682.45   131.4 2675.55   228.5 2638.45   319.5 2609.72
   347.6 2608.94   375.6  2614.1   403.3 2614.54   430.2 2605.88   483.1 2601.56
   507.4 2600.21  523.31 2601.61   534.6 2604.32   569.2 2602.29   589.8  2605.1
   610.4 2603.22   680.7 2604.64   708.2  2602.5   759.7 2605.25  1395.5 2603.37
  1430.4 2605.55  1512.4 2604.75    1776 2608.16  1971.6 2613.46  1992.1 2613.38
  2005.7  2610.3    2034 2615.24  2082.8 2636.36  2101.2 2642.23  2149.6 2650.37
#Mann= 7 ,-1,0
       0     .12       0   483.1     .04       0  523.31     .08       0
  638.63     .07       0  878.63     .05       0 1829.38     .07       0
 1959.38     .08       0
Bank Sta=483.1,523.31
XS Rating Curve= 0 ,0
Exp/Cntr(USF)=0,0
Exp/Cntr=0.3,0.1

Type RM Length L Ch R = 1 ,59131   ,345.6,357.9,363.5
XS GIS Cut Line= 3
2304848.38856814528932.6573312542305250.12151989529639.707326332
2304643.50476275530230.254765402
#Sta/Elev= 30
       0 2681.82    83.4 2678.83   155.7 2679.27   179.2 2674.96   208.5 2662.99
   226.3 2653.57   240.8 2643.87     249 2635.05   278.9  2608.8     295  2600.5
   308.8 2598.76   355.2 2599.14   361.52600.481   368.6 2602.26   396.2 2603.06
   454.9 2602.01   479.1 2603.85   548.1 2604.38     631 2603.37  1016.9 2604.37
  1058.9 2606.18  1435.6 2611.92  1446.7 2611.81  1457.9 2609.19  1497.3 2615.97
  1534.1 2634.33  1586.3 2663.86  1610.5  2675.8  1641.1 2687.46  1659.8  2691.3
#Mann= 8 ,-1,0
       0     .05       0      30      .1       0     295     .04       0
   361.5      .1       0     450     .05       0 1383.21     .07       0
 1483.21     .08       0 1623.21      .1       0
Bank Sta=295,361.5
XS Rating Curve= 0 ,0
Exp/Cntr(USF)=0,0
Exp/Cntr=0.3,0.1

Type RM Length L Ch R = 1 ,58773   ,345.3,366.2,382
XS GIS Cut Line= 3
2304619.52130553529110.0063601332304873.36393124529925.843287814
2304601.77705817530186.299877929
#Sta/Elev= 30
       0 2678.17    70.3 2677.16     129 2674.98     150 2673.68   163.8 2671.34
   179.3 2666.13     196 2658.25   204.2 2653.24   221.2 2639.63   250.5 2606.65
   258.7  2601.7   271.4 2599.22     284 2598.22   313.3 2598.39   317.5 2599.35
   325.3 2602.45   338.3 2603.12   384.5 2601.31   426.4 2601.24   501.8 2603.52
   594.1 2603.94  1027.4 2611.81  1047.2 2608.85  1064.1 2614.44  1073.1  2616.2
  1083.3  2620.7  1113.5 2636.16  1188.6  2678.2  1211.2 2689.58  1230.7 2697.85
#Mann= 7 ,-1,0
       0      .1       0     250     .07       0   271.4     .04       0
   317.5     .07       0     460     .05       0 1014.42     .08       0
 1134.42      .1       0
Bank Sta=271.4,317.5
XS Rating Curve= 0 ,0
Exp/Cntr(USF)=0,0
Exp/Cntr=0.3,0.1

Type RM Length L Ch R = 1 ,58407   ,538.4,585,609.3
XS GIS Cut Line= 3
2304511.16187646529101.2204604782304388.15928129529262.295287482
2304326.65798371530102.813021119
#Sta/Elev= 30
       0 2677.33    24.9 2675.95    45.2 2672.89    95.6 2658.25   124.8 2644.82
   161.9 2623.43   181.1 2614.18   191.2 2610.27   217.6 2603.34   261.4  2602.6
   289.8 2604.04     358 2604.57     378  2602.7   398.1 2602.81   410.1 2600.67
   426.5 2599.67   446.2 2597.81   474.3 2597.95  475.96 2599.56   478.3 2602.32
   482.3 2603.22   542.5 2601.35   562.5 2605.14   702.9 2604.29   915.5 2606.97
   943.5 2614.73   951.5 2615.73   975.6 2625.04  1012.6 2633.02  1045.4 2641.83
#Mann= 6 ,-1,0
       0      .1       0     190     .08       0  392.67     .07       0
   426.5     .04       0  475.96     .07       0  982.67      .1       0
Bank Sta=426.5,475.96
XS Rating Curve= 0 ,0
Exp/Cntr(USF)=0,0
Exp/Cntr=0.3,0.1

Type RM Length L Ch R = 1 ,57822   ,757.4,775.1,774.6
XS GIS Cut Line= 2
2304484.80417749529095.3631940422303576.92787984529710.376169874
#Sta/Elev= 30
       0 2677.15    29.7 2674.82    50.7  2671.3    93.9 2659.83   142.9 2638.46
   189.2 2613.07   226.4 2598.83   276.1 2601.54   307.1 2600.51     339 2602.01
   396.9 2601.71   407.9 2600.51   527.4 2602.08   538.1 2601.78   559.5 2597.86
   585.4 2597.88   609.5 2601.13   648.2 2601.52   701.3 2599.39   706.1 2600.57
   713.2 2598.71     742 2596.99   753.4 2598.52   764.1 2602.66     837 2600.92
   860.7 2604.93   944.7 2605.37   991.2 2611.58  1021.4 2613.36  1096.6 2614.43
#Mann= 8 ,-1,0
       0      .1       0     250     .08       0     490     .07       0
     620     .08       0   713.2     .04       0   753.4     .08       0
     850     .07       0     970     .05       0
Bank Sta=713.2,753.4
XS Rating Curve= 0 ,0
Exp/Cntr(USF)=0,0
Exp/Cntr=0.3,0.1

Type RM Length L Ch R = 1 ,57047   ,767.5,758.5,752.4
XS GIS Cut Line= 2
2304418.85335555528823.5733112672303217.81480347529277.889705212
#Sta/Elev= 30
       0  2677.8   105.5 2677.06   131.2 2674.64   152.3 2669.91   186.8  2656.3
   203.9 2647.06   226.7 2632.61   242.2 2616.81   255.2 2605.37   259.5 2602.63
     268 2599.94   288.8 2600.51   302.2  2598.1   357.8 2599.03   383.5 2597.57
   426.2 2599.21   541.7 2598.26   558.8 2599.87   592.4 2600.48   836.8 2600.19
   845.4  2599.3   850.4  2597.3   858.2 2595.92   875.1  2596.2   879.6 2597.35
   884.5 2602.39   892.4 2604.11  1095.5 2608.93  1161.8 2612.84  1284.1 2617.26
#Mann= 6 ,-1,0
       0      .1       0     260     .08       0     680     .07       0
   850.4     .04       0   879.6     .07       0     890     .05       0
Bank Sta=850.4,879.6
XS Rating Curve= 0 ,0
Exp/Cntr(USF)=0,0
Exp/Cntr=0.3,0.1

Type RM Length L Ch R = 1 ,56288   ,400.8,394.6,386.3
XS GIS Cut Line= 2
 2304341.3011498528512.5651836112303172.77649572529010.432830713
#Sta/Elev= 30
       0 2671.98    31.7 2668.13    66.4 2659.46    75.1 2657.97    83.2 2658.16
    98.9 2660.95   114.3 2662.59     123 2662.72   131.7 2661.71   178.2 2650.39
   205.6 2645.49     236 2635.12   253.4  2627.5   262.1 2621.54   266.6 2617.51
   279.5 2601.99   283.8 2597.76   287.9 2596.14     294 2595.23   306.2 2595.03
   325.42596.013   344.7 2598.97   368.9  2600.2   427.3  2598.6   588.2    2601
   692.5 2600.58   749.1 2601.25  1153.4 2610.54    1230 2613.75  1270.2 2613.85
#Mann= 6 ,-1,0
       0      .1       0   287.9     .04       0   325.4      .1       0
     370     .07       0     390      .1       0     500     .05       0
Bank Sta=287.9,325.4
XS Rating Curve= 0 ,0
Exp/Cntr(USF)=0,0
Exp/Cntr=0.3,0.1

Type RM Length L Ch R = 1 ,55894   ,392,387.7,382.8
XS GIS Cut Line= 3
2304178.51899647528104.6108980812303713.62951894528400.049225196
2303173.54098355528989.325899925
#Sta/Elev= 30
       0 2676.69    51.4 2676.34    92.8 2674.94   116.5 2673.05   130.7 2669.94
   163.9 2658.12   187.6 2650.57   197.1 2646.76   224.8 2631.09   239.7 2616.95
   258.7 2599.94   267.52594.812   272.9 2593.75   297.7 2593.66   306.4 2593.75
   312.2 2594.59   320.3 2595.06   329.8 2598.25   338.3 2599.21   353.5 2598.34
   378.8 2598.66   403.8 2600.05     431 2600.53   538.3 2599.19     612 2600.94
     697 2600.81   742.3 2602.31     920 2602.92  1203.8 2610.18  1350.2 2612.66
#Mann= 5 ,-1,0
       0     .12       0     110      .1       0   267.5     .04       0
   312.2      .1       0     350     .05       0
Bank Sta=267.5,312.2
XS Rating Curve= 0 ,0
Exp/Cntr(USF)=0,0
Exp/Cntr=0.5,0.3

Type RM Length L Ch R = 1 ,55506   ,110.8,109.9,108.2
XS GIS Cut Line= 4
2304005.62286378527710.3847927542303724.85358299527942.767543995
2303765.36371972528146.0951743582303222.58710184528772.526564157
#Sta/Elev= 30
       0 2628.72    12.3 2623.35    23.2  2628.3    29.5 2629.19    79.7 2625.23
   102.4 2629.35   117.3 2632.24   129.9 2632.94   142.1 2632.61   164.9 2629.69
     220  2621.6   261.5 2617.03   270.1 2613.48   291.2 2598.41     303 2594.52
   312.7 2592.32   334.2 2592.55   341.1 2594.65     355 2598.19   436.3 2596.58
   501.5 2597.75   525.8 2599.87   697.6 2598.76   747.8 2599.74  1122.1 2601.77
  1141.9 2602.03  1252.5 2604.47  1306.6 2605.82    1383 2607.99  1400.7 2608.67
#Mann= 14 ,-1,0
       0     .06       0   102.4     .12       0   164.9      .1       0
   291.2     .05       0     303     .04       0   341.1     .05       0
   501.5     .06       0   697.6     .05       0   747.8     .06       0
  1122.1     .05       0  1141.9     .06       0  1252.5     .05       0
  1306.6     .06       0    1383     .05       0
#XS Ineff= 3 ,-1
       0     235  2602.5   411.6  790.892600.162  934.55 1299.67 2605.85
Permanent Ineff=
       F       F       F
Bank Sta=303,341.1
XS Rating Curve= 0 ,0
Exp/Cntr(USF)=0,0
Minor Loss Coefficient=0
Exp/Cntr=0.5,0.3

Type RM Length L Ch R = 1 ,55396   ,197.6,191.7,187.4
XS GIS Cut Line= 4
 2303904.8388761527655.3626480142303624.06959531527887.745399255
2303664.57973204528091.0730296182303121.80311416528717.504419417
#Sta/Elev= 30
       0 2653.16    30.2 2638.67      53 2627.38    99.5 2609.72   115.8 2612.14
   178.5 2605.99   214.8 2605.06   230.6 2594.84     235 2592.69   260.5 2592.38
   274.5 2592.66   280.2 2594.75   286.4 2598.08   341.6  2598.3     476  2598.6
   504.6 2601.02   545.4 2599.75   633.1 2598.91   682.4 2602.81     738 2600.57
   802.2  2600.6     843 2600.56   933.7 2601.89   993.9 2602.18  1066.8 2602.07
  1143.5 2602.65  1193.8 2602.96  1293.2 2605.06  1322.2 2606.06  1400.7 2608.23
#Mann= 15 ,-1,0
       0     .12       0    30.2     .06       0   230.6     .04       0
   280.2      .1       0   341.6     .06       0   545.4     .05       0
   802.2     .06       0     843     .05       0   933.7     .06       0
   993.9     .05       0  1066.8     .06       0  1143.5     .05       0
  1193.8     .06       0  1293.2     .05       0  1322.2     .06       0
#XS Ineff= 2 , 0
             225  2602.5     285            2600
Permanent Ineff=
       F       F
Bank Sta=230.6,280.2
XS Rating Curve= 0 ,0
Exp/Cntr(USF)=0,0
Minor Loss Coefficient=0
Exp/Cntr=0.5,0.3

Type RM Length L Ch R = 1 ,55205   ,216,219.5,223.1
XS GIS Cut Line= 2
2303817.53709582527448.1243557432302747.30258519528510.411580406
#Sta/Elev= 30
       0 2610.59    18.5 2607.54    52.6 2605.24    75.2 2607.54    92.1 2607.17
   103.4 2604.95   115.1 2600.64   120.7 2600.34   148.5 2603.07   204.8 2602.74
   238.6 2598.15   255.5 2598.41   264.8 2594.97   272.4 2592.51   300.6 2592.41
   311.9    2595   319.5 2597.64   330.8 2596.76   347.9 2597.87   363.8 2597.02
   512.5 2597.63   557.9 2600.07   691.8 2598.71   782.4  2600.8    1069 2599.35
    1184 2600.41  1219.3 2604.46  1247.5 2613.08  1257.5 2614.96  1507.9 2618.33
#Mann= 9 ,-1,0
       0     .12       0      50      .1       0   264.8     .04       0
   311.9      .1       0     460     .05       0     740     .07       0
     880     .05       0    1020     .07       0    1160     .05       0
#XS Ineff= 2 , 0
                         1064.42         2604.76
Permanent Ineff=
       F       F
Bank Sta=264.8,311.9
XS Rating Curve= 0 ,0
Exp/Cntr(USF)=0,0
Minor Loss Coefficient=0
Exp/Cntr=0.3,0.1

Type RM Length L Ch R = 1 ,54985   ,663.9,650,638.4
XS GIS Cut Line= 3
2303664.78687638527323.5400970022302792.05417735   528061.555668
2302715.90971367528477.421584991
#Sta/Elev= 30
       0 2674.63    53.2 2671.45   115.1 2657.94   177.6 2635.61   203.1 2621.28
   231.3 2597.57   244.1 2596.44   250.3 2594.18   262.7 2592.16   281.3 2592.43
   293.7 2594.37   299.9  2595.7   330.9 2596.53   356.4 2595.47   367.7 2598.59
   374.2 2598.99   424.5 2597.17   464.2 2599.51   516.7  2598.7   547.7 2600.22
   648.7 2598.75   807.7 2599.59   981.3 2598.43  1006.1 2600.07  1037.1 2611.65
  1064.2 2617.12    1130 2617.65  1268.6 2618.31  1419.1 2617.17  1565.7 2618.44
#Mann= 11 ,-1,0
       0      .1       0      90     .12       0     100      .1       0
   250.3     .04       0   293.7      .1       0     360     .05       0
     490     .03       0     540     .05       0     620     .03       0
     690     .07       0    1130     .05       0
Bank Sta=250.3,293.7
XS Rating Curve= 0 ,0
Exp/Cntr(USF)=0,0
Exp/Cntr=0.3,0.1

Type RM Length L Ch R = 1 ,54335   ,689.9,673.8,658.1
XS GIS Cut Line= 3
2303181.56239537526813.9579170272302554.83488667527768.692346175
2302279.54336415527929.767173179
#Sta/Elev= 30
       0 2678.51      39 2677.85    82.7 2674.62   104.4 2671.02   133.3 2662.56
   145.7 2657.46     157 2650.82   211.3 2604.87   221.2 2598.52   230.3 2594.77
   238.3 2591.75     267 2591.64   276.6 2594.31   295.1 2595.99   314.9    2594
   323.2 2594.22   338.4 2596.81   357.9 2595.12   396.1 2595.94     418 2593.91
   456.8 2595.73   482.3 2595.77   505.5 2598.08   745.7 2597.38   956.6 2599.19
   994.1 2604.45  1005.7 2604.94  1205.4 2608.25  1298.1  2612.3    1461 2617.36
#Mann= 6 ,-1,0
       0      .1       0     210     .08       0   230.3     .04       0
   276.6     .08       0     910      .1       0 1312.06     .05       0
Bank Sta=230.3,276.6
XS Rating Curve= 0 ,0
Exp/Cntr(USF)=0,0
Exp/Cntr=0.3,0.1

Type RM Length L Ch R = 1 ,53661   ,609.5,603.2,597.9
XS GIS Cut Line= 2
2302516.76265483526453.7360311822302194.61300082 527894.62357456
#Sta/Elev= 30
       0 2668.86    36.3 2671.47    77.1  2672.4   126.5 2672.77   138.8 2670.73
   155.2 2659.41   167.5 2648.22   171.6 2643.66     188 2619.95     201 2603.37
  211.42 2594.84   216.7 2591.72   220.8  2590.8   253.6 2590.51   261.12594.431
   265.8 2595.72   302.7 2596.62   345.1 2594.43   376.5 2596.69   454.4 2596.23
   528.2  2598.1   653.1 2597.24   683.9 2598.39  1028.4 2598.25  1058.6  2599.9
  1075.3 2604.86  1112.2 2611.39  1151.2 2614.26  1229.1 2616.03  1476.5 2617.27
#Mann= 8 ,-1,0
       0      .1       0  211.42     .04       0   261.1     .08       0
     650      .1       0     850     .08       0    1050      .1       0
    1250     .05       0    1450      .1       0
Bank Sta=211.42,261.1
XS Rating Curve= 0 ,0
Exp/Cntr(USF)=0,0
Exp/Cntr=0.3,0.1

Type RM Length L Ch R = 1 ,53058   ,379.9,387.2,395
XS GIS Cut Line= 4
 2302030.6095406526483.0223633652301866.60608038 526623.59675784
2301802.17614958527399.6845606762302051.10997313527865.337242378
#Sta/Elev= 30
       0 2666.81    50.6 2665.73    66.4 2664.61    82.7 2662.41   102.5 2657.51
   128.1 2648.12     156 2636.69   179.1 2625.04   207.5 2607.89   229.6 2595.79
  239.32 2591.34   241.7 2590.01   245.7  2589.5   285.8 2589.46   297.6 2591.36
   317.9  2596.5   362.1 2594.03   416.1 2596.64   470.5 2597.14     627 2596.77
   663.1 2595.94   755.4  2597.2   916.5 2597.36  1015.1 2599.87  1100.8 2604.19
  1177.6 2606.24  1248.6 2610.84  1309.4 2613.02  1363.8 2614.47  1522.8 2615.88
#Mann= 6 ,-1,0
       0      .1       0      20     .12       0  239.32     .04       0
   297.6     .12       0  486.01     .08       0  976.01      .1       0
Bank Sta=239.32,297.6
XS Rating Curve= 0 ,0
Exp/Cntr(USF)=0,0
Exp/Cntr=0.3,0.1

Type RM Length L Ch R = 1 ,52671   ,889.5,920.9,944.1
XS GIS Cut Line= 4
2301849.10795706526093.2400968062301557.44769865526287.450793531
2301404.95853754526919.8943528792301022.72084774527313.298999187
#Sta/Elev= 30
       0  2636.6    14.3 2628.48    21.5 2627.81    43.2 2635.43    63.6 2638.78
   136.2 2643.42   182.4 2650.57     227 2655.21   245.3 2652.37   259.7 2654.52
   268.9 2652.62   294.3 2640.08   317.4 2620.56     341  2603.1   356.4 2596.15
   555.1 2594.23   611.4 2596.22   628.1  2593.8   636.1 2590.44   644.6 2589.31
   677.2 2589.42   681.4 2590.63   684.4 2593.36   689.6 2595.11   841.8 2594.33
     883 2596.25  1064.1 2595.19  1234.4 2598.24  1386.7 2610.15  1549.5  2626.5
#Mann= 9 ,-1,0
       0      .1       0     190     .12       0     280      .1       0
   360.4     .12       0   490.4      .1       0   560.4     .08       0
   628.1     .04       0   684.4     .08       0 1230.97     .12       0
Bank Sta=628.1,684.4
XS Rating Curve= 0 ,0
Exp/Cntr(USF)=0,0
Exp/Cntr=0.3,0.1

Type RM Length L Ch R = 1 ,51750   ,570.8,567.6,560.2
XS GIS Cut Line= 2
2301721.61790665525935.5609364492300235.20598518526743.044169469
#Sta/Elev= 30
       0 2658.58    83.6 2653.85   162.6 2638.34   183.7 2632.04   217.6 2610.66
   238.2  2599.7   256.6 2597.62   353.3 2594.96   575.2 2595.49   670.8 2592.22
     689 2593.79   739.1 2591.87   893.9 2594.14   971.2 2592.41  1008.9 2594.55
  1089.6 2594.05  1107.8 2592.09  1148.8 2594.25  1194.3 2592.48  1217.1 2594.08
  1230.7 2593.03  1245.3 2589.11  1267.1 2588.34  1277.1 2588.95  1321.8 2601.97
  1394.8 2611.27  1517.5 2623.36  1558.5 2631.05  1617.6 2637.24  1691.6  2648.2
#Mann= 9 ,-1,0
       0     .06       0      10      .1       0     340     .08       0
  1245.3     .04       0  1277.1     .08       0    1350     .05       0
    1370     .08       0    1460     .05       0    1570      .1       0
#XS Ineff= 2 , 0
          356.21  2603.4
Permanent Ineff=
       F       F
Bank Sta=1245.3,1277.1
XS Rating Curve= 0 ,0
Exp/Cntr(USF)=0,0
Exp/Cntr=0.3,0.1

Type RM Length L Ch R = 1 ,51182   ,573.7,540.4,502
XS GIS Cut Line= 2
2301525.25760861525502.2556389422300080.46522094526377.591567507
#Sta/Elev= 30
       0 2667.27    75.7 2668.72   113.6 2665.83   142.7 2650.22   183.5  2633.2
   244.5 2614.17   279.6 2596.18   291.2 2593.13   679.4 2593.55   702.8 2590.84
   772.9 2592.34   791.7  2590.2   833.7 2589.88     946  2592.9   955.3  2589.6
   978.3 2587.53   996.5 2589.42  1007.7 2591.39  1047.8  2592.1  1070.9 2589.28
  1086.3 2590.91  1128.4 2590.05  1142.4 2591.59  1156.2 2596.22  1179.8 2600.21
  1438.7 2603.65  1525.9 2607.74  1558.7 2610.98  1619.3  2622.2  1689.3 2630.94
#Mann= 13 ,-1,0
       0     .12       0      10      .1       0     120     .12       0
     240      .1       0     390     .08       0     700     .07       0
     810     .08       0   955.3     .04       0   996.5     .08       0
    1040     .07       0    1150     .08       0    1160     .05       0
    1620      .1       0
#XS Ineff= 2 , 0
          367.58  2604.9
Permanent Ineff=
       F       F
Bank Sta=955.3,996.5
XS Rating Curve= 0 ,0
Exp/Cntr(USF)=0,0
Exp/Cntr=0.3,0.1

Type RM Length L Ch R = 1 ,50642   ,285.7,273.8,258.7
XS GIS Cut Line= 3
 2300493.7279084525049.9445085682300360.31239513525895.994104951
 2300067.4490733526335.289087688
#Sta/Elev= 30
       0 2634.98    15.4 2631.32    47.8 2627.85    88.1 2625.66   112.6 2618.47
   130.1 2620.83   153.1 2608.04   168.6 2603.36   189.5  2601.1   245.5 2598.06
   294.8 2597.66   319.1 2594.15   367.7    2592   420.3 2590.47   533.7 2591.46
  543.39 2589.38   549.9 2587.03   570.2 2586.78   586.4 2589.34   614.7 2591.68
     635 2589.87   707.9 2589.85     716 2591.42   732.2 2590.33   773.7 2598.95
   941.1 2606.05  1229.6 2609.28  1260.6 2612.66  1324.2  2624.9  1384.5 2630.26
#Mann= 8 ,-1,0
       0      .1       0     470     .08       0  543.39     .04       0
   586.4     .08       0   986.5     .05       0  1066.5     .08       0
  1106.5     .05       0  1336.5      .1       0
Bank Sta=543.39,586.4
XS Rating Curve= 0 ,0
Exp/Cntr(USF)=0,0
Exp/Cntr=0.3,0.1

Type RM Length L Ch R = 1 ,50368   ,210.6,247.2,286.1
XS GIS Cut Line= 4
2300415.63102258525056.4525823872300161.81614367 525625.90904149
2300236.65899258526003.3773229542300047.92485185526322.272940052
#Sta/Elev= 30
       0  2628.3    62.1 2619.54    70.9 2617.06    79.6 2612.49    88.4    2615
    97.1 2614.46   101.5 2613.11   115.2 2599.99   145.3 2597.14   224.6 2594.69
   250.4 2595.71   263.6 2594.32   368.7 2593.31   381.8 2590.25     400 2589.77
   708.4 2591.13   721.3 2588.26   728.7 2586.67   745.1 2586.61   761.4 2586.69
   769.62588.222   781.8 2590.04     794 2596.69   805.2 2598.24    1006 2606.22
  1120.9 2606.98  1211.4 2609.47  1251.2 2614.34  1310.7 2625.64  1378.8 2631.12
#Mann= 10 ,-1,0
       0      .1       0     390     .08       0     420     .06       0
     500     .08       0   721.3     .04       0   769.6     .08       0
  903.46      .1       0 1003.46     .08       0 1118.28     .05       0
 1348.28      .1       0
#XS Ineff= 2 , 0
          297.65 2599.11
Permanent Ineff=
       F       F
Bank Sta=721.3,769.6
XS Rating Curve= 0 ,0
Exp/Cntr(USF)=0,0
Exp/Cntr=0.5,0.3
